HEC-RAS study BACKCREEK.prj: BACKCREEK

--- BACKCREEK.g01 (geometry) --- (continued)

Type RM Length L Ch R = 1 ,63984.1 ,447.9,427.4,406.9
XS GIS Cut Line= 3
     2378607.615      374839.706      2378802.06      374791.095
     2379819.421      375148.734
#Sta/Elev= 30
       0   522.8      59  500.55   121.8  472.37   145.4  463.03   188.6  452.59
   236.4  444.87   296.3  429.58   344.2  425.71   396.1  425.51   448.1  422.49
     508  421.64   563.9  421.63   719.6  425.95   723.6  424.92   735.6  414.16
   739.6   413.5   819.5  413.95   827.5  417.18   835.5  416.75  847.69418.4288
   855.4   422.6   859.4  423.05   911.4  423.11   923.4  424.68   959.3  432.92
  1007.2  451.53 1016.56 453.155  1071.1  458.27  1115.1  460.09  1278.8  457.74
#Mann= 5 ,-1 , 0
       0     .12       0   735.6    .045       0   819.5     .04       0
  847.69     .12       0 1016.56     .06       0
Bank Sta=735.6,819.5
XS Rating Curve= 0 ,0
Exp/Cntr=0.3,0.1

Type RM Length L Ch R = 1 ,63556.7 ,680.8,669.1,657.4
XS GIS Cut Line= 3
     2378680.532      375534.151     2378847.198      375461.234
      2379833.31      375284.151
#Sta/Elev= 30
       0  570.62    55.4  562.52      83  556.66    98.9  552.03   118.6  543.22
   237.8  484.26   257.8  471.46   297.7  439.38   313.6  429.83   325.6  424.96
   345.6   422.5   393.5  422.23   445.4  424.49   465.3  422.73   485.3   423.2
   493.3  422.22  507.86417.3133   517.2   413.7   521.2   413.5     617  413.72
  632.45421.1103   748.7  428.39   828.6  424.82   848.5  429.46   868.5  439.17
   896.4  449.31   916.4  454.64  926.96454.9684  1032.1  458.79  1183.8  456.81
#Mann= 6 ,-1 , 0
       0     .12       0  507.86     .04       0   517.2    .045       0
     617     .04       0  632.45     .12       0  926.96     .06       0
Bank Sta=517.2,617
XS Rating Curve= 0 ,0
Exp/Cntr=0.3,0.1

Type RM Length L Ch R = 1 ,62887.6 ,653.4,642.6,631.9
XS GIS Cut Line= 2
     2379027.754      376176.512     2380006.921      375617.484
#Sta/Elev= 30
       0   543.9      44  535.42      72  526.25      88   519.5   191.9  463.63
   223.9  443.54   247.9  424.55   263.9  420.16  277.27418.5674   291.9  413.68
   295.9   413.5   373.7413.8905  376.23414.6075   387.8  423.26   399.8  424.38
   415.8  422.35   455.8  424.61   483.8  423.99   527.8   427.3   563.8  422.91
   599.7  422.43   631.7  425.87   679.7  425.49   723.7  427.05   775.7  434.97
   819.6  448.07   843.6  454.04  851.09454.0428   955.6  457.04  1127.5  458.37
#Mann= 6 ,-1 , 0
       0     .12       0  277.27     .04       0   291.9    .045       0
   373.7     .04       0  376.23     .12       0  851.09     .06       0
Bank Sta=291.9,373.7
XS Rating Curve= 0 ,0
Exp/Cntr=0.3,0.1

Type RM Length L Ch R = 1 ,62245   ,680.6,678.6,676.7
XS GIS Cut Line= 2
     2379394.772      376850.978     2380271.508       375943.86
#Sta/Elev= 30
       0  465.42   127.8  465.13   223.6  460.77  250.73457.3501  258.82456.0756
   315.4     446   347.3  434.15   375.3  428.66   399.2  426.21  448.85 425.125
   459.1  422.83   467.1  414.44  470.94413.5376   471.1   413.5  572.28413.6794
  576.32415.2234   582.9  421.07   598.8  422.02   614.8   426.6   650.7  427.68
  741.57425.3338  792.66425.5442   898.3  428.08   950.2  431.99   962.1   434.6
   994.1  446.31    1050  452.32  1161.8  454.73  1217.6  452.51  1261.6  448.45
#Mann= 9 ,-1 , 0
       0     .12       0  250.73     .06       0  258.82     .12       0
  448.85     .04       0  470.94    .045       0  572.28     .04       0
  576.32     .12       0  741.57    .016       0  792.66     .12       0
Bank Sta=470.94,572.28
XS Rating Curve= 0 ,0
Exp/Cntr=0.3,0.1

Type RM Length L Ch R = 1 ,61566.3 ,669.8,659.7,649.7
XS GIS Cut Line= 4
     2379749.976       377186.06     2380013.474        377199.6
     2380604.143      376429.116     2380843.726      376377.033
#Sta/Elev= 30
       0  461.61  174.54450.6578  257.87446.5047  266.03445.7491  385.41436.0234
   467.6  426.06   519.5  426.22   575.5  422.77   607.4  416.33   631.4  419.21
   695.3  420.39  739.47416.0943   767.2   413.3   831.2   413.1   837.2 413.265
  838.33413.3582   851.2  420.08   859.1  422.04   887.1  417.26   899.1  417.34
   903.1  418.46   915.1  426.98     967  423.61 1016.41424.4306  1046.9  422.92
 1058.65425.2813 1248.29  447.63 1396.52459.8477 1402.49460.2297  1479.9  464.88
#Mann= 14 ,-1 , 0
       0     .12       0  174.54    .016       0  257.87     .12       0
  266.03     .06       0  385.41     .12       0  739.47     .04       0
   767.2    .045       0   837.2     .04       0  838.33     .12       0
 1016.41    .016       0 1058.65     .12       0 1248.29     .06       0
 1396.52     .08       0 1402.49     .06       0
Bank Sta=767.2,837.2
XS Rating Curve= 0 ,0
Exp/Cntr=0.3,0.1

Type RM Length L Ch R = 1 ,60906.6 ,886.1,882.4,878.6
XS GIS Cut Line= 3
     2380193.673      378341.342     2380485.339      377952.454
     2381145.062      376563.565
#Sta/Elev= 30
       0  504.03   119.5  501.88   207.2  495.13     263  487.81   374.5  464.04
  421.82457.3338  462.72452.7867   597.9  442.36   737.7  440.65  964.29428.5838
 1036.29424.2563 1053.35423.9896  1137.1  424.59  1236.9  421.16  1316.8  423.52
 1418.55420.8058 1485.36423.4905  1532.5  423.69  1552.4  418.67  1600.4  417.17
  1612.4  413.09  1680.3  413.09  1692.2  417.17 1693.32417.6348 1700.98421.7706
  1708.2  425.32  1724.2  424.16 1745.23427.2261    1812  454.38  2023.7  492.25
#Mann= 13 ,-1 , 0
       0     .12       0  421.82    .016       0  462.72     .06       0
  964.29     .12       0 1036.29     .08       0 1053.35     .12       0
 1418.55     .06       0 1485.36     .12       0  1600.4    .045       0
  1692.2     .04       0 1693.32     .12       0 1700.98    .016       0
 1745.23     .12       0
Bank Sta=1600.4,1692.2
XS Rating Curve= 0 ,0
Exp/Cntr=0.3,0.1

Type RM Length L Ch R = 1 ,60024.2 ,546.1,550.4,554.9
XS GIS Cut Line= 4
       2381391.3      378643.513     2381409.789      378146.541
     2381881.921      376951.685     2382081.404      376846.638
#Sta/Elev= 30
       0  477.71   21.09476.4278    43.8  475.13   57.19472.0403   97.16466.8895
   143.2  455.63     183  449.36  305.29441.4922     629  438.33  716.15431.9855
   828.5  424.25  881.53422.6119  994.28421.0458 1037.07419.9947  1287.3  422.28
 1349.67419.6615    1427   422.9    1435  420.97  1450.9   413.3  1454.9  412.78
  1590.6  413.14  1598.5     417  1614.5  429.09  1666.4  443.85  1682.3  444.88
  1722.2   454.7  1865.1  477.19  1888.9  484.23  1936.3  502.95  2007.5  520.54
#Mann= 12 ,-1 , 0
       0     .06       0   21.09     .12       0   57.19    .016       0
   97.16     .12       0  305.29     .06       0  716.15     .12       0
  881.53     .08       0  994.28     .12       0 1037.07     .06       0
 1349.67     .12       0  1450.9    .045       0  1590.6     .12       0
Bank Sta=1450.9,1590.6
XS Rating Curve= 0 ,0
Exp/Cntr=0.3,0.1

Type RM Length L Ch R = 1 ,59473.8 ,645.4,643.3,640.8
XS GIS Cut Line= 3
     2381829.837      378540.227     2381838.518      378240.748
     2382411.435      377073.213
#Sta/Elev= 30
       0  448.28   31.81443.3199   72.04439.4744   183.8  434.57   311.6  440.71
   407.3  440.92   495.1  434.91   606.8  422.54  657.81421.1041  670.89421.2758
   726.5  419.14  747.78421.2614   830.2  422.08   949.9  418.46  1009.7  421.93
 1102.88422.0811 1133.29423.1715 1153.06410.8324  1157.3  410.64  1229.1  410.99
 1231.08411.4899  1249.1  419.12    1281   419.5    1285  421.62  1296.9   438.3
  1304.9  442.12  1500.4  465.19  1520.4  471.89  1580.2  503.97  1600.1  510.55
#Mann= 11 ,-1 , 0
       0     .12       0   31.81    .016       0   72.04     .12       0
  657.81     .06       0  670.89     .12       0  747.78     .06       0
 1102.88     .12       0 1133.29     .04       0 1153.06    .045       0
  1229.1     .04       0 1231.08     .12       0
#XS Ineff= 2 , 0
       0   367.4                       0
Permanent Ineff=
       F       F
Bank Sta=1153.06,1229.1
XS Rating Curve= 0 ,0
Exp/Cntr=0.3,0.1

Type RM Length L Ch R = 1 ,58830.5 ,646.2,644.9,643.5
XS GIS Cut Line= 3
     2382302.758      378734.658     2382459.178      378518.526
     2382936.608      377411.755
#Sta/Elev= 30
       0  468.14    59.7   467.6   131.4  464.15  304.75444.4295   318.7  441.73
   334.8440.8285   470.4  428.89   550.2  426.62   586.1  424.08  688.77422.3922
   797.6   422.5  838.81420.1309  891.02418.6424  1021.1  421.08 1065.68419.1439
    1085   418.6    1105   420.3 1110.83417.9893  1116.9  413.27  1124.9  410.95
  1128.9  410.64  1252.6  410.81  1256.6  416.86  1260.6  426.08  1264.6  432.28
  1268.6  435.76  1280.6  442.04  1296.5  445.23  1384.3  446.96  1472.2  446.42
#Mann= 10 ,-1 , 0
       0     .12       0  304.75    .016       0   334.8     .12       0
  688.77     .06       0  838.81     .12       0  891.02     .06       0
 1065.68     .12       0 1110.83     .04       0  1124.9    .045       0
  1252.6     .12       0
Bank Sta=1124.9,1252.6
XS Rating Curve= 0 ,0
Exp/Cntr=0.3,0.1

Type RM Length L Ch R = 1 ,58185.6 ,537.8,527.4,517.1
XS GIS Cut Line= 4
     2383149.112      379016.776     2383070.987      378639.172
     2383570.119      377480.318     2383622.203      377384.832
#Sta/Elev= 30
       0  461.01   53.21461.4671  116.74 461.114  148.61461.2211   381.6  460.92
   449.5   453.8  521.97438.2234  558.92431.9088   649.1  423.13  723.58422.2959
  842.13  421.53   904.7  423.22   912.7  420.14  920.11  411.57   924.6  410.64
  1000.5  411.35 1006.43414.8997  1040.4  419.33  1232.1  418.19  1248.1  422.41
  1347.9   423.2  1411.8  417.85  1479.7  419.98  1495.6  418.61  1511.6  412.48
  1539.6  412.03  1551.6  415.15  1575.5  432.75  1623.4     444  1756.1  485.38
#Mann= 11 ,-1 , 0
       0     .06       0   53.21     .12       0  116.74     .06       0
  148.61     .12       0  521.97    .016       0  558.92     .12       0
  723.58     .06       0  842.13     .12       0  920.11    .045       0
  1000.5     .04       0 1006.43     .12       0
Bank Sta=920.11,1000.5
XS Rating Curve= 0 ,0
Exp/Cntr=0.3,0.1

Type RM Length L Ch R = 1 ,57658.2 ,718.9,735.9,752.8
XS GIS Cut Line= 3
     2383544.247      378878.769     2383717.858      378757.241
     2383862.923       377281.22
#Sta/Elev= 30
       0  460.49  239.34 448.274  240.71448.2884  310.97446.4323  362.56445.5165
   387.8   444.7   463.8  421.74  522.71420.6196   611.7  421.33   620.7416.4125
  626.76410.4167   671.6  409.32   680.9410.0563  717.08415.9763   743.6  412.08
   759.6  415.15   783.6  413.27   907.5  417.11   971.5  423.56  1207.3  423.28
  1275.3  419.32  1359.2   420.3  1379.2  411.51  1419.2  411.83  1463.2  452.55
  1547.1  497.26  1559.1  500.63  1607.1  531.14  1651.1  547.08    1695  551.56
#Mann= 10 ,-1 , 0
       0     .06       0  239.34     .12       0  240.71    .016       0
  310.97     .06       0  362.56     .12       0  522.71     .06       0
   620.7     .04       0  626.76    .045       0   680.9     .04       0
  717.08     .12       0
Bank Sta=626.76,680.9
XS Rating Curve= 0 ,0
Exp/Cntr=0.3,0.1

Type RM Length L Ch R = 1 ,56922.3 ,587.3,601.3,615.3
XS GIS Cut Line= 3
     2383965.254      378861.408     2384164.907      378709.498
     2384794.247      377672.171
#Sta/Elev= 30
       0  450.91   37.86449.4458   167.2  446.66   374.6  450.14  462.09442.4635
   486.4  436.99   554.2  414.65     654  414.44  682.12411.3623   709.9  409.04
   717.8   408.5  775.52409.2617   785.7  416.69   809.6  418.97   965.3  418.06
   993.2  409.37  1005.2  410.09  1021.2  415.52  1037.1  427.05    1089  449.92
  1136.9  475.71  1212.7  525.18  1228.7  542.25  1264.6  570.88  1272.6  579.85
  1296.6  615.52  1336.5  647.12  1356.4  670.41  1384.4  692.62  1464.2  741.49
#Mann= 6 ,-1 , 0
       0     .12       0   37.86     .06       0  462.09     .12       0
  682.12     .04       0   709.9    .045       0  775.52     .12       0
Bank Sta=709.9,775.52
XS Rating Curve= 0 ,0
Exp/Cntr=0.3,0.1

Type RM Length L Ch R = 1 ,56321.1 ,689.9,697.9,705.7
XS GIS Cut Line= 2
     2384147.546      379160.887     2385262.997      378297.171
#Sta/Elev= 30
       0  445.42   115.9   439.1  212.27442.1035  307.06 448.004   411.6  450.05
  552.61442.1079   607.5  437.57   703.4  418.42   859.2  419.94  961.56416.5586
   971.1  414.78   983.1  408.39   987.1  408.17  1051.1  408.56 1062.21409.2935
    1083  409.67    1095  414.71    1183   484.1  1206.9  511.58  1214.9  527.44
  1222.9  540.13  1234.9  554.83  1246.9   566.6  1250.9  573.08  1266.9   606.6
  1270.9  611.78  1306.8  629.48  1318.8   641.3  1338.8  670.43  1410.8  720.11
#Mann= 8 ,-1 , 0
       0     .06       0  212.27     .12       0  307.06     .06       0
  552.61     .12       0  961.56     .04       0   983.1    .045       0
  1051.1     .04       0 1062.21     .12       0
Bank Sta=983.1,1051.1
XS Rating Curve= 0 ,0
Exp/Cntr=0.3,0.1

Type RM Length L Ch R = 1 ,55623.2 ,600.4,612.2,624
XS GIS Cut Line= 3
     2384462.914      379541.934     2385283.476      379148.514
     2385679.664      378956.894
#Sta/Elev= 30
       0  447.27   16.96 446.492   259.4   447.9  395.82437.3516  472.63430.3499
   582.7  419.92  689.43 419.332  724.48419.4784  799.73419.3323   862.1  420.81
   874.1  417.96  885.96409.3744     886  409.35     898  408.17   973.4  408.88
  976.95411.6845   993.3  420.22    1021  447.45  1036.9  468.71  1060.7   486.2
  1064.6  495.88  1072.6  522.88  1088.4  544.66  1108.2  557.29  1120.1  570.68
  1147.9  587.39  1175.6   612.3  1270.8   679.7  1318.4   711.9  1350.1  729.15
#Mann= 11 ,-1 , 0
       0     .12       0   16.96     .06       0  395.82     .12       0
  472.63     .06       0  689.43     .12       0  724.48     .07       0
  799.73     .12       0  885.96     .04       0     886    .045       0
   973.4     .04       0  976.95     .12       0
Bank Sta=886,973.4
XS Rating Curve= 0 ,0
Exp/Cntr=0.3,0.1

Type RM Length L Ch R = 1 ,55011   ,402.6,405.2,407.7
XS GIS Cut Line= 3
     2384593.651      379832.759     2385731.747       379677.38
     2386005.185      379581.894
#Sta/Elev= 30
       0  443.59   155.6  440.42   219.4  442.39   267.2  439.37  323.79430.9162
     351  428.04   378.9  427.17  405.31424.6169  448.21423.4298   538.4  418.15
   570.3  419.16  626.68418.5324   792.7  420.17   881.4  422.31   901.4   419.1
   905.4  416.83   913.3  409.26   917.3  408.17   997.1  408.17 1003.06409.0462
 1011.65414.8439    1021  420.76    1037  435.12  1068.9  459.69  1100.8  481.28
  1220.1  554.99  1251.8  576.47  1267.7  585.46  1339.1   633.9  1438.3     695
#Mann= 9 ,-1 , 0
       0     .06       0  323.79     .12       0  405.31     .06       0
  448.21     .12       0  626.68     .06       0   792.7     .12       0
   913.3    .045       0 1003.06     .04       0 1011.65     .12       0
Bank Sta=913.3,1003.06
XS Rating Curve= 0 ,0
Exp/Cntr=0.3,0.1

Type RM Length L Ch R = 1 ,54605.8 ,462,465.2,468.6
XS GIS Cut Line= 2
     2384702.034      380162.039     2385970.462      380076.685
#Sta/Elev= 30
       0  466.87      48   457.8      72  454.41   147.9  450.27   195.9  443.71
   211.9  439.84   259.9  431.11   315.8  425.98   415.8  422.89   443.8   420.6
   499.7  419.25   591.7  419.93   615.7  417.71  677.82 419.489   739.6  420.09
   787.6  418.69  824.76418.9872   855.5  420.64   859.5  419.99   863.5  417.32
  869.21411.7096  873.69408.8973   879.5  408.17  956.74408.9066  959.71410.3223
   971.5  417.68  1007.4  455.66  1019.4  465.41  1167.4  568.88  1271.3   644.6
#Mann= 7 ,-1 , 0
       0     .12       0  677.82     .06       0  824.76     .12       0
  869.21     .04       0  873.69    .045       0  956.74     .04       0
  959.71     .12       0
Bank Sta=873.69,956.74
XS Rating Curve= 0 ,0
Exp/Cntr=0.3,0.1

Type RM Length L Ch R = 1 ,54140.6 ,511.2,515,518.6
XS GIS Cut Line= 2
     2384695.839      380546.114     2386062.973      380575.181
#Sta/Elev= 30
       0  503.26      36  502.05      68   497.8      88  493.55     132  479.96
   227.9  443.52   243.9  438.24   263.9  434.03   323.9  427.95   403.8  424.98
   451.8  419.54   479.8  418.52  543.12419.3205   607.8  418.48  717.21  419.54
   843.7  421.69   851.6   418.3   859.6  409.46   867.6  408.17   951.6  408.17
  956.65409.7353  962.21414.2372   971.6  420.72   991.6  439.68  1051.6  486.35
  1083.6  514.78  1151.5  563.26  1183.5  588.92  1251.5  630.36  1367.4  692.38
#Mann= 6 ,-1 , 0
       0     .12       0  543.12     .08       0  717.21     .12       0
   859.6    .045       0  956.65     .04       0  962.21     .12       0
Bank Sta=859.6,956.65
XS Rating Curve= 0 ,0
Exp/Cntr=0.3,0.1

Type RM Length L Ch R = 1 ,53625.6 ,526.2,533.1,539.9
XS GIS Cut Line= 3
     2384639.074      380965.654     2385909.698      381118.352
     2386052.928      381144.394
#Sta/Elev= 30
       0  489.51      48     481     100  467.71     172  457.11     196  454.42
     240  455.47   327.9  442.23   347.9  436.52   387.9  419.14  472.94418.7256
  632.86  417.62  703.14418.6643   779.9  421.27   799.8  417.72   811.8  407.87
   815.8  407.76  838.39407.8183   855.8  415.52  868.18415.8053   875.8  414.33
   883.8  408.68   955.8  409.31  977.54418.3615   995.8  419.49  1023.8  441.18
  1091.8  477.06  1287.6  593.56  1382.1   643.8  1401.7   656.8  1425.3  664.06
#Mann= 9 ,-1 , 0
       0     .12       0  472.94     .08       0  632.86     .06       0
  703.14     .12       0  838.39     .04       0  868.18     .12       0
   883.8    .045       0   955.8     .04       0  977.54     .12       0
Bank Sta=883.8,955.8
XS Rating Curve= 0 ,0
Exp/Cntr=0.3,0.1

Type RM Length L Ch R = 1 ,53092.6 ,571.7,576.8,581.9
XS GIS Cut Line= 3
     2384505.857      381310.106     2385692.685      381678.248
      2385935.74      381695.609
#Sta/Elev= 30
       0  468.58   131.8  457.87   235.7  457.16   359.6  441.91   395.6  441.14
   411.5  437.92   455.5  418.96  513.16417.1112  680.81417.1921  758.05417.3112
   823.1  418.38   843.1  414.53     855  407.73     859  407.35   960.7  408.17
   970.9  416.52   977.8 418.667  1034.8  418.09  1058.8  419.24  1070.8  421.63
  1102.8  436.89  1174.7  455.68  1214.6  470.35  1226.6  473.12  1286.6  502.39
  1362.4  536.04  1382.4   547.8  1410.4  553.52  1434.4  566.31  1486.3  583.69
#Mann= 7 ,-1 , 0
       0     .12       0  513.16     .08       0  680.81     .06       0
  758.05     .12       0     855    .045       0   960.7     .04       0
   977.8     .12       0
Bank Sta=855,960.7
XS Rating Curve= 0 ,0
Exp/Cntr=0.3,0.1

Type RM Length L Ch R = 1 ,52515.7 ,634.9,640.5,646.1
XS GIS Cut Line= 2
     2384355.829      381737.506     2385679.664      382355.331
#Sta/Elev= 30
       0  452.72   287.4  442.67   399.2  428.21   423.1  418.98   435.1  416.86
  502.75 416.455   582.8  418.09  653.01 417.044  746.84418.1644   818.3  416.34
   826.2  413.25   830.2  409.09   834.2   407.2   838.2  406.96   918.1  406.49
  928.33406.9313  941.01412.3179     950  415.71  1013.8  418.09  1037.8  422.94
  1065.7  425.94  1205.4  436.24  1261.3  443.15  1285.3  448.03  1317.2  457.75
  1349.1  469.64  1385.1  486.26    1401  489.03    1421  498.86  1460.9  512.86
#Mann= 7 ,-1 , 0
       0     .12       0  502.75     .08       0  653.01     .06       0
  746.84     .12       0   838.2    .045       0  928.33     .04       0
  941.01     .12       0
Bank Sta=838.2,928.33
XS Rating Curve= 0 ,0
Exp/Cntr=0.3,0.1

Type RM Length L Ch R = 1 ,51875.2 ,590.9,593,595.1
XS GIS Cut Line= 3
     2384126.636      382181.018     2385202.233      382893.526
     2385588.518      382828.421
#Sta/Elev= 30
       0  441.49   111.8  445.25   179.8  445.76   299.6  432.97   355.5  414.89
  397.25 415.374   472.2415.2793  503.57 415.108  648.54416.8996   878.8  419.57
   886.8  418.34   890.8  414.88   894.7  408.64  898.57405.8923   902.7  405.71
   978.6  406.04   990.6   411.6  997.12412.9728  1018.6  416.96  1034.5  425.94
  1142.4  467.69  1198.3  480.99 1233.01486.8646 1251.78488.7732  1274.2  489.37
  1298.2  494.65  1390.1  507.74  1438.1  512.84    1566  518.65  1681.9  527.75
#Mann= 10 ,-1 , 0
       0     .12       0  397.25     .08       0   472.2     .12       0
  503.57     .06       0  648.54     .12       0  898.57    .045       0
   978.6     .04       0  997.12     .12       0 1233.01    .016       0
 1251.78     .12       0
Bank Sta=898.57,978.6
XS Rating Curve= 0 ,0
Exp/Cntr=0.3,0.1

Type RM Length L Ch R = 1 ,51282.2 ,694.5,701.6,708.6
XS GIS Cut Line= 3
     2383652.585      382497.679     2384742.164      383310.192
     2384720.462      383566.269
#Sta/Elev= 30
       0   437.7      76  433.82   179.9  434.88  224.11438.0863   271.8  440.34
  310.26439.0315  316.32438.9061  343.82437.5582   371.8  435.01   403.8   428.1
   431.7  426.77  500.37417.0463   519.7  414.56  666.37413.9923  695.61  414.51
  823.06414.7768  1095.3  420.46  1123.3  418.79  1127.3  416.64  1135.3  407.19
  1139.3  405.71  1235.2  407.12  1243.2   413.7 1253.14 415.923  1287.2  435.17
  1319.2  445.56  1442.2  464.83 1506.83469.4539 1591.49 471.511  1616.2  472.06
#Mann= 14 ,-1 , 0
       0     .12       0  224.11     .06       0  310.26     .12       0
  316.32     .06       0  343.82     .12       0  500.37     .07       0
  666.37     .12       0  695.61     .06       0  823.06     .12       0
  1135.3    .045       0  1235.2     .04       0 1253.14     .12       0
 1506.83    .016       0 1591.49     .12       0
Bank Sta=1135.3,1235.2
XS Rating Curve= 0 ,0
Exp/Cntr=0.3,0.1

Type RM Length L Ch R = 1 ,50580.7 ,712.6,703.8,695.1
XS GIS Cut Line= 3
     2383396.678      382915.227     2384282.094      383878.769
     2384481.747       383900.47
#Sta/Elev= 30
       0  446.05  158.52433.0078   243.4  430.56   311.2  423.41     379  420.54
   430.9  420.04  495.16414.1459   570.5  412.06   609.1413.2223   873.5 416.042
   941.5  417.83   965.5  412.82   981.4  405.88   985.4  405.71  1077.2  405.97
  1081.2  407.94  1089.2  418.19 1094.54419.1024  1121.1  418.64    1133  419.99
  1172.9  440.78  1224.8  462.83  1260.7   463.9  1276.7   467.1  1320.4  466.75
    1344  468.71  1367.6  468.34 1480.98472.0374 1509.29472.6649  1509.4  472.67
#Mann= 10 ,-1 , 0
       0     .06       0  158.52     .12       0  495.16     .07       0
   609.1     .06       0   873.5     .12       0   981.4    .045       0
  1077.2     .04       0 1094.54     .12       0 1480.98     .06       0
 1509.29     .12       0
Bank Sta=981.4,1077.2
XS Rating Curve= 0 ,0
Exp/Cntr=0.3,0.1

Type RM Length L Ch R = 1 ,49876.8 ,691.1,684.6,678.1
XS GIS Cut Line= 3
     2382841.122      383579.289     2383809.004      384234.671
     2383960.914       384217.31
#Sta/Elev= 30
       0  440.42    79.8  435.46   147.6  434.62   271.3  423.07   355.1  420.23
     379  413.77   402.9  411.32   418.9  406.47   434.8  405.06  436.54405.1862
   458.8  407.45  475.36411.9491   510.6  415.53     758  417.39     766  415.91
     774   406.9  776.99405.5813   841.8  405.48   857.7  408.55  894.01409.7702
   905.6  413.86   929.5  415.95  1073.2  414.12  1085.1  417.66  1109.1  431.67
    1129  438.45  1196.3  444.85  1237.5451.3577 1267.01457.9337  1321.8  466.16
#Mann= 8 ,-1 , 0
       0     .12       0  436.54     .04       0  475.36     .12       0
  776.99    .045       0   841.8     .04       0  894.01     .12       0
  1237.5    .016       0 1267.01     .12       0
Bank Sta=776.99,841.8
XS Rating Curve= 0 ,0
Exp/Cntr=0.3,0.1

Type RM Length L Ch R = 1 ,49192.2 ,638.2,601,563.9
XS GIS Cut Line= 3
     2382470.431      384282.069     2383379.316      384694.741
     2383665.775      384620.956
#Sta/Elev= 30
       0  553.76      16  552.55    35.9  543.45   103.8  505.87   163.7  470.44
   195.6  453.15   231.6  436.45   267.5  424.55   307.4  417.67   343.4  407.06
  368.89408.4096   395.3     406   423.2  406.94  433.59412.5018   463.2   416.4
     567  416.23   642.8  414.04   646.8   413.3   654.8  405.79   658.8   405.1
   730.7  405.65   738.7  412.08  753.05413.5891   774.6  413.23   802.5  416.72
   822.5  421.07   850.4  432.38   882.4   436.5  1130.1  444.13    1294  445.25
#Mann= 6 ,-1 , 0
       0     .12       0  368.89     .04       0  433.59     .12       0
   654.8    .045       0   730.7     .04       0  753.05     .12       0
Bank Sta=654.8,730.7
XS Rating Curve= 0 ,0
Exp/Cntr=0.3,0.1

Type RM Length L Ch R = 1 ,48591.2 ,724.6,696.1,667.3
XS GIS Cut Line= 3
     2382385.393      385580.158     2383414.039      384937.796
     2383574.629      384829.289
#Sta/Elev= 30
       0  517.09    20.7517.7551   37.78517.7189    79.8     514   89.87510.4395
   135.6  488.71   175.5  445.68   211.4  417.67   223.4  413.41   263.3  414.04
  274.57407.7307   287.2  404.57   315.2  404.11  345.49409.6019   454.8  407.06
   518.6  414.64     738  413.89   797.9  411.13   805.8  405.38  863.14 405.538
   864.4405.8687  879.54409.0082   945.5  412.06  1014.4426.8912  1061.2  432.93
  1105.5434.5163 1146.53434.8845 1238.98437.9981 1296.84 440.433  1406.6  443.45
#Mann= 15 ,-1 , 0
       0     .06       0    20.7     .08       0   37.78    .016       0
   89.87     .12       0  274.57     .04       0  345.49     .12       0
   805.8    .045       0  863.14     .04       0   864.4     .08       0
  879.54     .06       0  1014.4     .12       0  1105.5    .016       0
 1146.53     .06       0 1238.98     .12       0 1296.84     .06       0
Bank Sta=805.8,863.14
XS Rating Curve= 0 ,0
Exp/Cntr=0.3,0.1

Type RM Length L Ch R = 1 ,47895.1 ,474.6,464.8,455.2
XS GIS Cut Line= 3
     2383266.469      386022.866     2383518.205      385814.533
     2383726.539      385033.283
#Sta/Elev= 30
       0  520.64    43.8  517.64    71.7  514.56   107.6  509.88   131.5  505.05
     259  471.67   326.8  451.96   342.7  445.33   362.6   439.1  382.07429.2336
   390.5  423.42   402.4   413.2   418.4  404.41   470.2  403.87   533.9  403.87
   541.8  404.64   553.8  410.15   577.7  412.44   593.6  411.06   613.5  410.98
   625.5  409.53   645.4  412.55   677.3  412.91   709.1   410.9   836.6  418.83
   884.4  422.84     976  436.58 1009.33440.1197 1049.94 441.822  1135.3  443.48
#Mann= 6 ,-1 , 0
       0     .12       0  382.07     .04       0   418.4    .045       0
   541.8     .12       0 1009.33    .016       0 1049.94     .06       0
Bank Sta=418.4,541.8
XS Rating Curve= 0 ,0
Exp/Cntr=0.3,0.1

Type RM Length L Ch R = 1 ,47430.4 ,786.3,786.4,786.6
XS GIS Cut Line= 4
     2384165.895       386494.12     2384012.223      386237.132
     2384008.657      385185.192     2383999.976      385085.366
#Sta/Elev= 30
       0  496.52    47.9  496.71   235.6  488.88   323.4  481.28   367.4  475.53
   431.4  463.38   559.4  434.35   619.4  417.92   651.4  415.54   742.6 414.788
   747.4  413.32   751.4  406.69  753.84404.7014   759.4  403.05   811.4  403.05
   819.4  404.92   871.4  406.04   883.4  411.28   891.4  412.76   907.4  411.22
   967.4   411.7  1027.4  409.84  1051.4  411.33  1135.4  411.21  1219.4  421.14
  1271.4  432.98 1361.12440.6628 1392.32442.0765 1451.25 443.211  1451.6  443.22
#Mann= 7 ,-1 , 0
       0     .12       0   742.6     .04       0  753.84    .045       0
   819.4     .12       0 1361.12    .016       0 1392.32     .12       0
 1451.25     .06       0
Bank Sta=753.84,819.4
XS Rating Curve= 0 ,0
Exp/Cntr=0.3,0.1

Type RM Length L Ch R = 1 ,46643.9 ,594.2,602.2,610.2
XS GIS Cut Line= 3
     2384559.872      386461.234     2384611.955      385228.595
     2384373.071      385045.422
#Sta/Elev= 30
       0  466.53    67.9  463.19   119.8  455.72   163.7  466.18   195.6  469.06
   331.4  462.43   371.3  455.96     535   415.7     571  412.24   626.8   413.7
   706.7  409.73   770.6  409.63   798.5  403.62   830.5  408.43   898.4  409.99
   922.3  412.89 1054.22411.7167    1070  410.38    1082  403.34    1090  402.23
  1149.9  403.94  1161.9  410.75  1173.8   421.8  1209.8  432.09 1254.98438.0036
 1330.78436.0372  1372.4  430.67 1396.84430.6158 1439.64431.7006  1534.8  438.43
#Mann= 8 ,-1 , 0
       0     .12       0 1054.22     .04       0    1082    .045       0
  1149.9     .12       0 1254.98    .016       0 1330.78     .12       0
 1396.84    .016       0 1439.64     .12       0
Bank Sta=1082,1149.9
XS Rating Curve= 0 ,0
Exp/Cntr=0.3,0.1

Type RM Length L Ch R = 1 ,46041.7 ,956.8,957.6,958.3
XS GIS Cut Line= 4
     2384782.596      386516.893     2384954.837      386318.005
      2385261.51      385138.191     2385215.254      384850.991
#Sta/Elev= 30
       0  464.33    95.7  480.91  190.05489.6926   263.1  492.14  347.76486.3397
     383   483.3     423  467.08   486.9  448.49   554.9  419.83   578.8  412.73
   598.8  410.04   698.8  410.64   730.7  406.14   762.7  408.27   778.7  403.28
   798.7  403.73   810.7  412.95   814.7  413.36   874.6  410.87 1215.63409.0574
 1237.08402.9191  1310.3   401.9  1318.3  403.28  1330.2  413.31  1350.2  414.98
  1398.2  410.44  1470.1  430.71 1528.34 434.482 1681.76443.1379    1773  455.09
#Mann= 8 ,-1 , 0
       0     .12       0  190.05    .016       0  347.76     .12       0
 1215.63     .04       0 1237.08    .045       0  1318.3     .12       0
 1528.34     .06       0 1681.76     .12       0
Bank Sta=1237.08,1318.3
XS Rating Curve= 0 ,0
Exp/Cntr=0.3,0.1

Type RM Length L Ch R = 1 ,45084.1 ,657.1,689.6,721.7
XS GIS Cut Line= 4
     2385358.483      386435.192     2385584.178      386383.109
     2385905.358      385172.171     2385992.164       384989.88
#Sta/Elev= 30
       0  477.59    36.4478.2125    91.8  476.59  254.48  447.26   302.6  438.93
   371.3  426.49   415.2  414.39   443.1  409.89     495  407.84   538.8  409.91
   550.8  406.39   562.8  399.85   618.6  400.14   646.6  406.23  647.48406.3224
   722.4   407.1   774.2  411.95  1113.4  411.63  1137.3  409.72 1228.47 411.939
  1284.9  409.86 1342.39414.5096  1368.7  427.09  1388.7  432.26  1424.6  432.46
    1524  446.75 1590.68451.0357 1622.27   451.8  1650.7   452.9  1686.3  460.91
#Mann= 11 ,-1 , 0
       0    .016       0    36.4     .12       0  254.48    .016       0
   302.6     .12       0   550.8    .045       0   646.6     .04       0
  647.48     .12       0 1228.47     .08       0 1342.39     .12       0
 1590.68    .016       0 1622.27     .12       0
Bank Sta=550.8,646.6
XS Rating Curve= 0 ,0
Exp/Cntr=0.3,0.1

Type RM Length L Ch R = 1 ,44394.5 ,640.9,650.4,660.3
XS GIS Cut Line= 3
     2385536.435      386478.595     2385866.296      386465.574
     2386803.796      385992.484
#Sta/Elev= 30
       0  460.56    83.5  443.56   111.7440.5231  151.78437.9209  188.14435.4183
   254.6  436.32   290.3  429.96   326.1  431.94   338.1  429.84   358.1  421.19
     418  409.73   685.5   411.7   701.4  408.92   741.4  408.18   753.4  400.36
   761.3  399.85   853.2  400.91   861.2  404.75   899.7407.1085  1012.9   402.3
  1028.9  403.05 1041.87409.1046  1084.8   411.4  1128.7  408.16  1152.6   415.8
  1220.5  463.24  1228.5   470.3  1240.5  487.05  1268.4  510.36  1380.2  589.93
#Mann= 8 ,-1 , 0
       0    .016       0   111.7     .12       0  151.78    .016       0
  188.14     .12       0   753.4    .045       0   853.2     .12       0
   899.7     .08       0 1041.87     .12       0
Bank Sta=753.4,853.2
XS Rating Curve= 0 ,0
Exp/Cntr=0.3,0.1

Type RM Length L Ch R = 1 ,43744.1 ,596.7,606.3,615.9
XS GIS Cut Line= 3
     2385727.407      387086.234      2386037.15      386896.875
     2386947.025       386708.63
#Sta/Elev= 30
       0  463.28    75.8  461.41   155.6  443.53   194.6 437.392  258.92432.1709
   287.2  430.77  349.95433.3446   398.9  428.14   446.8  420.27   578.4  409.98
  717.05409.9534  755.66410.5386   841.6   409.3   865.5  406.51   873.5  403.42
   905.4  406.99   961.2  407.07   973.2  400.66   981.1  399.85 1046.08400.7862
 1051.42403.7462  1060.9  409.14  1092.8  434.44  1116.7  457.54  1144.6  479.81
  1160.6  501.46  1168.6  509.16  1188.5  519.72  1232.4  549.72  1292.2  581.92
#Mann= 9 ,-1 , 0
       0     .06       0   194.6     .12       0  258.92     .06       0
  349.95     .12       0  717.05     .06       0  755.66     .12       0
   973.2    .045       0 1046.08     .04       0 1051.42     .12       0
Bank Sta=973.2,1046.08
XS Rating Curve= 0 ,0
Exp/Cntr=0.3,0.1

Type RM Length L Ch R = 1 ,43137.8 ,782.7,797.5,810.8
XS GIS Cut Line= 3
     2385729.557      387314.427     2386894.941      387372.692
     2387064.212      387481.199
#Sta/Elev= 30
       0  472.73      36  470.62   127.9  451.25   175.8  443.81   243.8  438.49
  306.14 436.718   351.6  436.05   459.5  417.66   559.4  409.89   667.3  408.01
  720.63410.1132   743.3  410.97  802.28408.8601  811.96409.4855  859.45411.2274
   939.1  409.87     951  407.58     975  406.01   984.7 400.736     991  399.85
  1066.9  400.77 1076.44409.9986  1090.9  425.65  1110.9  438.71  1130.9  447.46
  1158.8  456.58  1237.8  489.03    1289  504.93  1308.8  509.67  1367.9  515.65
#Mann= 9 ,-1 , 0
       0     .06       0  306.14     .12       0  720.63     .06       0
  802.28     .12       0  811.96     .06       0  859.45     .12       0
   984.7    .045       0  1066.9     .04       0 1076.44     .12       0
Bank Sta=984.7,1066.9
XS Rating Curve= 0 ,0
Exp/Cntr=0.3,0.1

Type RM Length L Ch R = 1 ,42340.3 ,189,191.5,195.7
XS GIS Cut Line= 6
     2385647.632      387580.201      2386425.41      387996.868
     2386616.382      388107.979      2386894.16      388222.562
     2387095.549      388222.562     2387539.994      388055.895
#Sta/Elev= 30
       0  470.74   89.18463.5103  135.55456.2072   154.3 453.366  239.72443.1389
  253.04442.0075   483.1  419.23  605.08420.6873  729.89420.6384  733.51420.4572
   767.3417.5378  790.51414.6035  851.14407.6471  875.44 401.812   929.7  400.78
   937.6  398.86  1016.5  400.79 1047.42407.4048  1162.6  418.87  1286.7411.7271
 1440.51439.3796  1526.2  446.53 1578.66434.8372  1613.2  427.63  1700.9  449.62
 1738.07440.7546  1804.6  443.13  1896.4  433.25  1992.1  445.79  2079.8  439.95
#Mann= 20 ,-1 , 0
       0     .06       0   89.18     .12       0  135.55     .06       0
   154.3     .12       0  239.72     .06       0  253.04     .12       0
  605.08     .08       0  729.89     .06       0  733.51     .08       0
   767.3     .12       0  790.51     .08       0  851.14     .06       0
  875.44     .12       0   929.7    .045       0  1016.5     .04       0
 1047.42     .06       0  1286.7     .12       0 1440.51     .08       0
 1578.66     .06       0 1738.07     .12       0
#XS Ineff= 2 , 0
       0     750            1160       0
Permanent Ineff=
       F       F
Bank Sta=929.7,1016.5
XS Rating Curve= 0 ,0
Exp/Cntr=0.3,0.1

Type RM Length L Ch R = 1 ,42148.8 ,448.5,451.3,454
XS GIS Cut Line= 6
     2385529.577      387705.201     2386307.355      388121.868
     2386440.215      388197.664     2386513.999      388336.552
     2386921.985      388575.268     2387171.551      388675.094
#Sta/Elev= 30
       0  471.67   81.88466.2368  304.34442.0813  338.15440.1941  375.74438.5546
  405.86436.4272   455.2  431.66     531  416.04  541.75417.2175     555  422.76
   574.9  423.56  593.94415.7808   610.9   409.5   634.8  408.38   838.4   407.7
  872.81400.3098   937.3  398.23   956.9  400.79  982.11400.7351  1141.5  409.53
  1224.4  407.35  1407.1  410.61  1466.7   419.5  1510.4  420.02 1634.08433.3686
  1678.3 439.221  1708.8  444.22  1736.4   444.1  1787.8   460.9  1934.1  494.21
#Mann= 13 ,-1 , 0
       0     .12       0   81.88     .06       0  304.34    .016       0
  338.15     .12       0  375.74     .06       0  405.86     .12       0
  541.75    .016       0  593.94     .12       0  872.81    .045       0
   956.9     .04       0  982.11     .12       0 1634.08     .06       0
  1678.3     .12       0
#XS Ineff= 2 , 0
       0     700            1290       0
Permanent Ineff=
       F       F
Bank Sta=872.81,956.9
XS Rating Curve= 0 ,0
Exp/Cntr=0.3,0.1

Type RM Length L Ch R = 1 ,41697.4 ,517.9,519.4,520.8
XS GIS Cut Line= 3
     2385442.771       388031.59     2386640.688      388871.868
     2386744.855      388941.312
#Sta/Elev= 30
       0  454.83      96  446.77   184.4442.2725   323.8     436   347.8  431.53
  388.45418.3593   407.8  416.48  419.78409.9226   427.8  406.13   439.8  404.47
   503.7   406.6   547.7  404.83   591.7  405.87   619.7  401.67   631.7  397.99
   711.6  397.99  719.82400.5224   731.6  409.72  757.76409.9424   919.5  407.54
  977.96409.4854  1010.2407.9822  1159.4  407.61 1283.04415.3759  1331.3  427.28
  1415.3  458.99  1443.2  466.92 1461.43469.4019  1486.7  472.92  1588.4  470.58
#Mann= 11 ,-1 , 0
       0     .06       0   184.4     .12       0  388.45    .016       0
  419.78     .12       0   619.7    .045       0  719.82     .04       0
  757.76     .06       0  977.96     .12       0  1010.2     .06       0
 1283.04     .12       0 1461.43     .06       0
Bank Sta=619.7,719.82
XS Rating Curve= 0 ,0
Exp/Cntr=0.3,0.1

Type RM Length L Ch R = 1 ,41178.1 ,577.7,589.9,602.1
XS GIS Cut Line= 3
     2384845.549      388370.131     2385390.292      388575.377
      2386362.91      389271.173
#Sta/Elev= 30
       0   448.8   191.4  436.45  304.16434.2268   382.8  431.07  427.95432.9612
  473.96434.7657   518.3  434.45   574.5429.6761  616.19424.7705   642.1  419.75
   658.1  419.83  666.92416.0143   690.1  402.47   710.1  402.03   722.1  398.62
   730.1  397.99   803.8398.5447  818.02 402.436   834.1  402.32   854.1  407.21
  926.13406.7807 1109.16  406.74    1346  404.81    1378  407.88 1479.31410.1793
    1514  412.45 1578.06422.5747    1622  429.06    1734  462.74    1778  471.78
#Mann= 14 ,-1 , 0
       0     .12       0  304.16     .06       0  427.95     .12       0
  473.96     .06       0   574.5     .12       0  616.19    .016       0
  666.92     .12       0   722.1    .045       0   803.8     .04       0
  818.02     .12       0  926.13     .06       0 1109.16     .12       0
 1479.31     .06       0 1578.06     .12       0
Bank Sta=722.1,803.8
XS Rating Curve= 0 ,0
Exp/Cntr=0.3,0.1

Type RM Length L Ch R = 1 ,40588.2 ,960.2,959,958.4
XS GIS Cut Line= 3
     2384817.771      388691.312     2385493.498      389619.223
     2385522.632      389667.875
#Sta/Elev= 30
       0  432.38      60  426.47     184  427.81     264  425.19   304.9421.7573
     336  418.61   347.5  415.65     384  406.97     408  398.23     412  397.63
  493.83398.8609     500  402.87  519.04402.0156   551.9  401.12   583.9   404.8
  669.39406.2123   751.9  405.68  848.45 409.021  916.54409.0492  953.42408.1786
  1003.9  407.89  1035.9  404.17  1055.9  405.62  1075.9  414.64  1091.9  424.93
  1111.9  440.83  1131.9  452.04  1174.3  467.05  1189.5   470.5  1204.6  470.93
#Mann= 10 ,-1 , 0
       0     .12       0   304.9    .016       0   347.5     .12       0
     408    .045       0  493.83     .04       0  519.04     .12       0
  669.39     .06       0  848.45     .12       0  916.54     .06       0
  953.42     .12       0
Bank Sta=408,493.83
XS Rating Curve= 0 ,0
Exp/Cntr=0.3,0.1

Type RM Length L Ch R = 1 ,39629.1 ,740.4,738.5,736.1
XS GIS Cut Line= 2
     2383712.737      388522.041     2384502.667      389780.722
#Sta/Elev= 30
       0  526.41      36  529.96   115.8  540.99   135.8  542.39   171.8  540.94
   215.7  534.93   251.7  525.87   283.6     514   435.4  441.34   447.4   434.6
   455.4  428.41  509.88419.4862  546.81416.2037   639.2  408.99     779  404.79
     787   402.8   794.9  398.14   802.9  397.37   922.8  398.29   930.8  405.57
  942.15 408.128  1094.5  404.39  1138.5  411.71  1186.4  437.77  1210.4  447.79
  1222.4  451.31  1234.4  453.08  1266.3  454.21 1344.96454.9907    1486  454.08
#Mann= 7 ,-1 , 0
       0     .12       0  509.88    .016       0  546.81     .12       0
   794.9    .045       0   922.8     .04       0  942.15     .12       0
 1344.96     .06       0
Bank Sta=794.9,922.8
XS Rating Curve= 0 ,0
Exp/Cntr=0.3,0.1

Type RM Length L Ch R = 1 ,38890.6 ,1622.2,1579.9,1537.6
XS GIS Cut Line= 2
     2382972.897      388802.367     2383938.431      389928.291
#Sta/Elev= 30
       0  502.49      36  503.33  210.69524.3972   255.9  527.34   311.8  527.48
   367.8  521.96   391.8  516.76   419.8   507.2   447.8  494.33   543.7  444.46
  564.71431.3107   591.7  430.15   605.6424.0627   663.6  408.73   679.6  398.26
   687.6  397.37  779.99397.5658   791.6  405.24  803.79407.2443  1007.5  405.19
  1059.4  407.41  1083.4  401.73  1111.4  406.83  1171.4  406.14  1203.4  403.61
  1247.4  407.54 1303.51418.0873  1339.3  421.77  1407.3  424.67  1483.2  424.86
#Mann= 8 ,-1 , 0
       0     .06       0  210.69     .12       0  564.71    .016       0
   605.6     .12       0   679.6    .045       0  779.99     .04       0
  803.79     .12       0 1303.51     .06       0
Bank Sta=679.6,779.99
XS Rating Curve= 0 ,0
Exp/Cntr=0.3,0.1

Type RM Length L Ch R = 1 ,37310.7 ,2689.3,2626.6,2563.5
XS GIS Cut Line= 2
     2381712.481      390620.075     2383981.834      390015.097
#Sta/Elev= 30
       0  485.23      12  483.84    67.9  468.24   171.8  451.15   239.6  442.78
   359.5  430.67   463.3  423.73   738.9   417.1   806.8  408.72   818.8  401.75
   834.8  397.04   850.8  396.06   914.7  397.62  916.42398.2736   930.7  402.35
   946.6  403.65  1158.3   402.9  1178.3   399.2  1206.3  402.46  1254.2  403.28
  1517.8  398.74  1565.7  405.89 1624.66404.6358 1688.47403.0863  1777.4  405.89
  1837.4  402.75 1881.51406.8878    2097   407.1  2252.8  415.42  2348.6  423.32
#Mann= 7 ,-1 , 0
       0     .12       0   834.8    .045       0   914.7     .04       0
  916.42     .12       0 1624.66     .06       0 1688.47     .12       0
 1881.51     .06       0
Bank Sta=834.8,914.7
XS Rating Curve= 0 ,0
Exp/Cntr=0.3,0.1

Type RM Length L Ch R = 1 ,34684.1 ,540.3,538.4,537
XS GIS Cut Line= 3
     2384347.897        391510.7     2384561.947      391099.027
     2384103.362      390015.097
#Sta/Elev= 30
       0  558.58   57.36 563.886  313.99561.7051  353.93559.5731     376  557.62
     404   549.9     460  539.54   503.9  545.83   531.8  546.51   547.8  543.45
   571.7  532.93   587.7  523.05  683.72458.4148  716.79436.3647   731.3  421.06
   759.2  401.24   779.2  399.43   819.1  402.34  849.96399.7606  858.62393.1968
   934.8  392.46  943.72393.3574   986.6  399.22  1070.4  397.84  1094.4  403.24
  1162.2  403.04    1238  407.64  1441.5  413.72  1529.2  422.38  1640.9   428.8
#Mann= 9 ,-1 , 0
       0     .12       0   57.36     .06       0  313.99    .016       0
  353.93     .12       0  683.72    .016       0  716.79     .12       0
  849.96     .04       0  858.62    .045       0  943.72     .12       0
Bank Sta=858.62,943.72
XS Rating Curve= 0 ,0
Exp/Cntr=0.3,0.1

Type RM Length L Ch R = 1 ,34145.7 ,936.3,943.5,950.7
XS GIS Cut Line= 2
     2385062.355      390902.454     2384632.875      389980.375
#Sta/Elev= 30
       0  481.76   139.6  450.73   163.6  440.25   171.5  440.48   211.4  451.22
   251.3  456.81   275.2  457.33   303.2  453.49   327.1  446.35     347  437.39
   382.9  412.88   406.9  402.31   438.8   396.7  474.68399.4902   510.6  392.93
   518.6  392.46   598.4  393.31   602.3  398.99   610.3  402.15   634.2  399.42
   658.2  402.88   674.1  402.76   690.1  401.37     706  397.07     726  402.28
   873.6  408.62   913.5  414.98   977.3  433.79  1009.1  438.03  1017.2  439.08
#Mann= 5 ,-1 , 0
       0     .12       0  474.68     .04       0   510.6    .045       0
   598.4     .12       0  1009.1     .06       0
Bank Sta=510.6,598.4
XS Rating Curve= 0 ,0
Exp/Cntr=0.3,0.1

Type RM Length L Ch R = 1 ,33202.2 ,1069.2,1078.3,1087.5
XS GIS Cut Line= 3
     2385618.119       390844.09     2385839.473      390653.118
     2385600.757      389702.597
#Sta/Elev= 30
       0  460.05   102.7  450.86  321.55427.9244   407.9  410.15   443.7  404.68
  574.63403.9328  688.86404.1989   734.6   403.1   778.4  404.31   798.3   403.1
   818.2  399.84  860.72399.5409     878  398.29     886  394.16   889.9  393.34
   925.8  393.44   933.8  392.12   937.7  392.04 1013.79392.1229  1017.4  392.89
  1025.4  399.86  1029.4  402.07  1033.4  402.76  1085.1  402.95  1140.9   398.9
  1152.9  403.89  1192.7  428.76  1224.6  446.25  1256.4  459.43  1272.4  463.88
#Mann= 7 ,-1 , 0
       0     .06       0  321.55     .12       0  574.63     .06       0
  688.86     .12       0  860.72     .04       0   933.8    .045       0
 1013.79     .12       0
Bank Sta=933.8,1013.79
XS Rating Curve= 0 ,0
Exp/Cntr=0.3,0.1

Type RM Length L Ch R = 1 ,32123.9 ,685.3,686,686.7
XS GIS Cut Line= 3
     2386399.981      391052.367     2386691.647      390776.325
     2386690.167      389381.416
#Sta/Elev= 30
       0  461.16  226.32455.3687   294.2  453.31   429.6  445.09  458.67441.4344
  471.65439.0486   537.5  416.94   569.4  411.14   661.4  402.85  792.55402.0144
  841.95402.6194  869.48401.4184  986.99403.4931 1004.55403.4486    1149  401.25
 1284.96403.0908  1391.9403.2112  1400.8  400.52 1411.06392.7126  1416.8  391.73
  1496.7  393.11  1508.7  395.42  1516.7  398.93  1528.7  408.82  1536.7  410.06
  1556.7  420.73  1604.6   438.6  1688.6  477.06 1737.09485.4075  1796.5  490.72
#Mann= 14 ,-1 , 0
       0     .06       0  226.32     .12       0  458.67     .06       0
  471.65     .12       0  792.55     .06       0  841.95     .12       0
  869.48     .06       0  986.99     .12       0 1004.55     .06       0
 1284.96     .12       0  1391.9     .04       0 1411.06    .045       0
  1496.7     .12       0 1737.09     .06       0
Bank Sta=1411.06,1496.7
XS Rating Curve= 0 ,0
Exp/Cntr=0.3,0.1

Type RM Length L Ch R = 1 ,31437.9 ,829.3,839.5,849.8
XS GIS Cut Line= 3
     2387345.549      390809.368      2387367.25      389476.902
      2387510.48      389225.166
#Sta/Elev= 30
       0  437.81  110.59 424.786   139.6  422.12   167.6  414.62   203.5  414.87
   243.4  405.63  365.09399.6497     395  402.11  447.34401.3822  470.12401.1602
  789.71400.7814   857.8  400.38   873.8  395.72   917.7  400.22  955.69395.4659
   969.6  393.38 1012.97393.5545  1025.4  397.09  1045.4     399 1125.11397.0418
 1154.02391.7776  1161.1  391.03  1232.9  391.65  1244.9  408.83  1260.8  419.69
  1332.6  430.51  1364.4  438.51  1447.7  471.12  1578.6   510.4  1622.3  520.66
#Mann= 11 ,-1 , 0
       0     .06       0  110.59     .12       0  365.09     .06       0
  447.34     .12       0  470.12     .06       0  789.71     .12       0
  955.69     .04       0 1012.97     .12       0 1125.11     .04       0
 1154.02    .045       0  1232.9     .12       0
Bank Sta=1154.02,1232.9
XS Rating Curve= 0 ,0
Exp/Cntr=0.3,0.1

Type RM Length L Ch R = 1 ,30598.3 ,648.5,652.9,657.3
XS GIS Cut Line= 4
      2387827.32      390783.326     2387938.138      390587.408
     2388213.605      389663.534     2388413.257      389576.729
#Sta/Elev= 30
       0   447.8    90.8  442.44   173.8  431.82     257  428.01   304.8   428.3
   336.6  426.38   388.4  416.86   444.2  398.77     484  397.82   507.9  399.38
  667.69399.3839  763.96400.2426   818.7  402.28   854.5   396.9   874.4  399.44
   902.3   399.2   918.3  397.96   934.1393.0185   946.2  391.35   954.1  390.78
  1057.7  391.52  1061.7  395.52  1077.6  419.65  1109.5  453.22  1129.4  468.15
  1173.2  494.22  1212.9  513.65    1300  548.81  1347.5  565.31  1406.9  581.58
#Mann= 6 ,-1 , 0
       0     .12       0  667.69     .06       0  763.96     .12       0
   934.1     .04       0   946.2    .045       0  1057.7     .12       0
Bank Sta=946.2,1057.7
XS Rating Curve= 0 ,0
Exp/Cntr=0.3,0.1

Type RM Length L Ch R = 1 ,29945.4 ,519.7,521.7,523.6
XS GIS Cut Line= 3
     2388381.023      390937.495     2388847.285      389863.187
     2389068.639      389802.423
#Sta/Elev= 30
       0  480.98      64  472.36   167.9   447.5   431.7  416.46   507.6   399.7
   563.6  398.53   579.6  395.94   615.5  399.56   655.5  398.07   707.5  401.26
   775.4   401.3   859.4  396.21   871.4   391.8  882.62392.5422   899.3  390.43
   907.3  389.36   979.3  389.38  985.19391.2936  985.46391.4812   995.3  401.14
  1031.2   424.9  1091.2  472.62  1139.2  513.96  1171.1  544.32    1183  551.65
  1206.8  571.02  1234.4  574.97    1274  587.78  1341.3  604.45  1400.7  615.29
#Mann= 5 ,-1 , 0
       0     .12       0  882.62     .04       0   899.3    .045       0
  985.19     .04       0  985.46     .12       0
Bank Sta=899.3,985.19
XS Rating Curve= 0 ,0
Exp/Cntr=0.3,0.1

Type RM Length L Ch R = 1 ,29423.8 ,495.2,510.4,525.7
XS GIS Cut Line= 3
       2388773.5      391091.486     2388942.771      390870.131
     2389363.778      390023.777
#Sta/Elev= 30
       0  466.94    79.6  452.29   191.1  440.81   338.5  423.14   442.2  409.03
     490  405.42     518  400.19   573.8  397.83  589.69389.7582   597.7  388.55
   635.6 389.035   669.5  395.74   689.5   398.1   709.4  397.08   745.3  398.79
   813.1  399.12  837.22396.4281     845  394.88  854.44389.7492     861  388.57
   928.8  389.22   948.7  398.99   968.7  417.12  1048.4  478.12  1076.4  503.73
  1092.3  520.81  1140.2  563.24  1164.1  572.04    1196  590.21  1223.9  603.13
#Mann= 6 ,-1 , 0
       0     .12       0  589.69     .04       0   635.6     .12       0
  837.22     .04       0  854.44    .045       0   928.8     .12       0
Bank Sta=854.44,928.8
XS Rating Curve= 0 ,0
Exp/Cntr=0.3,0.1

Type RM Length L Ch R = 1 ,28913.3 ,527.1,544.1,561.1
XS GIS Cut Line= 2
     2388981.834      391169.611     2389962.737      390336.277
#Sta/Elev= 30
       0  452.64   287.8  422.26   403.7  405.03   419.7  400.92   487.7  396.45
   515.6  398.78   595.6  399.95   631.6  398.58  642.38394.9188   651.5  388.69
   659.5  388.55   727.5  388.56  733.57390.2254   747.5  399.94   767.5  398.27
   779.4  396.28   787.4     390   795.4  388.55   839.4  388.67   855.4  398.16
   883.4   416.7   927.4  451.97   999.3  517.05  1015.3  533.14  1039.3  572.48
  1067.2  595.64  1123.2  629.98  1143.2  639.48  1187.2   653.7  1287.1  678.52
#Mann= 5 ,-1 , 0
       0     .12       0  642.38     .04       0  733.57     .12       0
   767.5    .045       0   855.4     .12       0
Bank Sta=767.5,855.4
XS Rating Curve= 0 ,0
Exp/Cntr=0.3,0.1
